--- 103_ras.prj (project) ---

Proj Title=103
Current Plan=p01
Default Exp/Contr=0.3,0.1
English Units
Geom File=g01
Flow File=f01
Plan File=p01
Y Axis Title=Elevation
X Axis Title(PF)=Main Channel Distance
X Axis Title(XS)=Station
BEGIN DESCRIPTION:
RFD model 103 exported to HEC-RAS
END DESCRIPTION:

--- 103_ras.p01 (plan) ---

Plan Title=Plan 01
Program Version=4.10
Short Identifier=Plan 01
Geom File=g01
Flow File=f01
Subcritical Flow
Calc Critical at every XS
Secant Critical Depth

--- 103_ras.f01 (steady flow) ---

Flow Title=Flow 01
Program Version=5.01
Number of Profiles= 5
Profile Names=10yr,25yr,50yr,100yr,500yr
River Rch & RM=103,47,11058.99
  152.79  273.01  390.09  531.35   954.4
River Rch & RM=103,47,10791.13
   156.5  279.79  399.97   545.1  980.53
River Rch & RM=103,47,10695.47
  168.23  301.23  431.28  588.74 1063.68
River Rch & RM=103,47,10599.82
  176.24   315.9  452.72  618.65 1120.89
River Rch & RM=103,47,10504.17
  212.46  382.39  550.18  755.02 1383.59
River Rch & RM=103,47,10408.51
  220.42  397.03  571.68  785.18 1442.08
River Rch & RM=103,47,10312.86
  226.53  408.29  588.23  808.41 1487.22
River Rch & RM=103,47,10217.21
  232.64  419.55  604.78  831.67 1532.47
River Rch & RM=103,47,10121.55
  252.16  455.55   657.8  906.22 1678.04
River Rch & RM=103,47, 10025.9
  255.21  461.18  666.09  917.89 1700.89
River Rch & RM=103,47,9930.246
  261.91  473.55  684.33  943.58 1751.24
River Rch & RM=103,47,9834.592
     285  516.27  747.38  1032.5 1926.14
River Rch & RM=103,47,9738.939
  288.64  523.01  757.35 1046.56 1953.88
River Rch & RM=103,47,9643.286
  295.32  535.37  775.62 1072.36 2004.83
River Rch & RM=103,47,9547.632
  299.56  543.23  787.24 1088.79 2037.31
River Rch & RM=103,47, 9454.37
   303.2  549.97  797.21 1102.88 2065.19
River Rch & RM=103,47,9361.108
  310.47  563.45  817.16 1131.08 2121.04
River Rch & RM=103,47,9157.904
  459.71  841.52 1230.54 1718.48 3300.32
River Rch & RM=103,47,9006.977
  476.47  872.87 1277.34 1785.29 3436.07
River Rch & RM=103,47,8894.798
  491.41  900.85 1319.14    1845 3557.67
River Rch & RM=103,47,8801.536
   493.2  904.21 1324.16 1852.17 3572.29
River Rch & RM=103,47,8608.103
  561.75 1032.84 1516.67 2127.71  4136.3
River Rch & RM=103,47,8414.671
  568.89 1046.26 1536.78 2156.54 4195.55
River Rch & RM=103,47,8221.238
  570.08 1048.49 1540.13 2161.34 4205.43
River Rch & RM=103,47,8027.806
  576.03 1059.67 1556.89 2185.38 4254.87
River Rch & RM=103,47,7834.373
  807.29 1496.13 2213.78 3131.29 6222.82
River Rch & RM=103,47,7640.941
  813.76 1508.39  2232.3 3158.05 6279.06
River Rch & RM=103,47,7447.508
  882.54 1638.79 2429.42 3443.23 6879.89
River Rch & RM=103,47,7279.075
  887.23  1647.7  2442.9 3462.76 6921.15
River Rch & RM=103,47,7134.203
  903.67 1678.89 2490.11 3531.14 7065.69
River Rch & RM=103,47,6797.881
  925.37 1720.11  2552.5 3621.57  7257.1
River Rch & RM=103,47, 6602.52
  937.09 1742.38 2586.24 3670.48 7360.74
River Rch & RM=103,47,6407.159
 1034.82 1928.29 2868.15 4079.74 8230.91
River Rch & RM=103,47,6211.799
 1041.25 1940.53 2886.74 4106.75 8288.51
River Rch & RM=103,47,6016.438
 1045.34 1948.32 2898.56 4123.94 8325.19
River Rch & RM=103,47,5821.078
 1051.18 1959.44 2915.46  4148.5 8377.61
River Rch & RM=103,47,5625.717
 1062.28 1980.58 2947.56 4195.18 8477.28
River Rch & RM=103,47,5430.356
 1066.95 1989.48 2961.08 4214.84 8519.28
Boundary for River Rch & Prof#=103,47,1
Up Type= 0
Dn Type= 2
Boundary for River Rch & Prof#=103,47,2
Up Type= 0
Dn Type= 2
Boundary for River Rch & Prof#=103,47,2
Up Type= 0
Dn Type= 2
Boundary for River Rch & Prof#=103,47,2
Up Type= 0
Dn Type= 2
Boundary for River Rch & Prof#=103,47,2
Up Type= 0
Dn Type= 2

--- 103_ras.g01 (geometry) ---

Geom Title=103
Program Version=4.10

River Reach=103,47
Reach XY= 30
1187478.29436839844230.496970698 1187629.4081125844240.157597587
1188124.93730086844088.3436663151188573.80174264843743.003877774
1188972.44899753843621.7100300941189151.68574533843481.101883635
1189154.00345796 843343.584031091189236.66868016843210.701609448
1189774.37892672842902.4452842031189921.21034959841940.397172838
1190179.20672297841528.0393201261190467.37615061841345.712271452
1190591.76026499840973.3324651421190852.11709532840865.172348917
1191132.84432653840572.367877245 1191004.5110248840362.367942974
1191062.84433246840068.2013615671190927.84436548  839839.8680996
1190791.17772198839254.0349432831190835.34437227839136.534976706
1191324.51089358839077.3683133421191436.17752343838937.368351489
1191891.17738295838699.8684084861192300.34393218838794.035035491
1192321.17727292839260.7015636711192380.34392422839329.868208185
1192812.01046199839255.7015509611193342.84364468 839437.36814858
1193549.51024696 839308.201514111193622.90941665839098.585157782

Type RM Length L Ch R = 1 ,11058.99,97.082200,97.082200,97.082200
XS GIS Cut Line= 6
1187454.27498482844479.1768504961187458.69652372844323.846088733
1187491.09111702844186.8136692321187498.31182662844136.377352915
 1187500.4052807844062.7108718741187495.63944425 843982.15811688
#Sta/Elev= 30
9749.078 400.8469754.308398.0343 9764.15390.79719770.712386.8118 9800.24372.7227
9813.364364.82539839.624352.31499849.492347.89189865.938342.21619915.411317.9806
9942.054309.01199952.044303.37929972.344290.34949975.753288.74499985.979284.7631
   10001281.746510006.43282.298510023.42286.660310033.61287.6496 10040.4290.0449
10067.04303.177710100.15315.7766 10146.1 335.41110169.07344.281110182.22 350.504
10208.51361.555210215.08365.088910238.09380.068710241.38381.5901 10250.9384.1523
#Mann= 3 , 0 , 0
9749.078  0.0734       09749.078  0.0734       0 10250.9  0.0734       0
#XS Ineff= 2 , 0
       0                               0
Bank Sta=9749.078,10250.9
Exp/Cntr=0.3,0.1

Type RM Length L Ch R = 1 , 10961.9,97.082300,97.082300,97.082300
XS GIS Cut Line= 6
1187593.91744286844494.9199123221187584.93371969844404.454339109
1187572.86436975844245.8338844651187570.47641452844218.775720682
1187563.32997051 844090.24585501 1187553.4669347 843994.66253186
#Sta/Elev= 30
 9749.01 335.6849789.868322.89659799.759322.00259812.947323.49449829.432324.4638
9836.025323.59599842.614321.73959852.485317.34869862.356312.09219885.388 301.995
9891.969 297.8669911.711284.10349924.872276.33479928.162275.61889957.775275.4581
10007.14273.740310013.72274.405310023.61276.360510063.04278.073910082.76280.7363
10092.62282.808910099.19285.837910112.33294.510710122.19299.492910138.62309.5509
10155.05315.611310184.73 328.78810194.63332.671110211.12338.197510250.98355.0991
#Mann= 3 , 0 , 0
 9749.01   0.076       0 9749.01   0.076       010250.98   0.076       0
#XS Ineff= 2 , 0
       0                               0
Bank Sta=9749.01,10250.98
Exp/Cntr=0.3,0.1

Type RM Length L Ch R = 1 ,10864.82,73.694900,73.694900,73.694900
XS GIS Cut Line= 3
1187779.07788716844427.7870977251187676.04434664844244.495851937
1187582.77187834844052.528097469
#Sta/Elev= 30
9769.578305.12629780.607302.43739799.425295.18089833.181280.80199837.062278.2404
9840.825276.52719885.989274.0131 9897.28272.10629908.571270.93779946.208270.7916
9949.972270.41849953.735270.46859961.263271.34179983.721270.382910023.84270.7683
10031.14270.013110038.44270.378910063.97273.504910093.15276.142310100.44276.3053
10107.74275.821110111.39 276.08110115.03277.577210123.19282.571210129.62287.3184
10140.57296.261110151.51303.201210162.45309.4154 10173.4315.129510193.27324.0343
#Mann= 3 , 0 , 0
9769.578  0.0846       09769.578  0.0846       010193.27  0.0846       0
#XS Ineff= 2 , 0
       0                               0
Bank Sta=9769.578,10193.27
Exp/Cntr=0.3,0.1

Type RM Length L Ch R = 1 ,10791.13,95.653400,95.653400,95.653400
XS GIS Cut Line= 3
1187818.12217623844386.5736815041187747.83373028 844227.88499333
1187660.86045647844023.244880676
#Sta/Elev= 30
9797.519293.88299806.017288.61489816.782279.9451 9820.37278.85539852.665276.2481
9884.959270.70449899.312   270.99906.488 270.4239913.665268.6727 9924.43263.7298
9928.018262.85789938.783261.66849978.207254.67589992.466253.945310017.42254.9586
10031.68257.134110045.94260.505810063.76261.060810088.72270.194510102.98276.8428
 10120.8283.033410127.93287.657110138.63292.589610149.32 299.63210152.88  300.98
10160.01302.567810172.19303.764910177.84305.407510184.97308.299310193.43309.5915
#Mann= 3 , 0 , 0
9797.519  0.0696       09797.519  0.0696       010193.43  0.0696       0
#XS Ineff= 2 , 0
       0                               0
Bank Sta=9797.519,10193.43
Exp/Cntr=0.3,0.1

Type RM Length L Ch R = 1 ,10695.47,95.653400,95.653400,95.653400
XS GIS Cut Line= 6
1187904.85629787844415.5873743341187853.37394808844244.625102928
1187839.93108897844205.7402702021187828.35525987844175.591776539
1187802.42143411844108.6820182961187748.86709337843938.722797725
#Sta/Elev= 30
9749.015313.15599773.725312.61069784.004310.36029794.283304.16819807.989297.4023
9818.268 285.9299821.694283.41089842.252279.88959869.663278.0973 9873.09  277.25
9886.795268.8305 9910.78267.10789917.833265.57669934.859258.44719973.102255.6248
9983.657253.49829997.731248.130410004.73247.331710032.88248.875410061.03 252.076
10075.05256.395810106.01268.729210154.17278.089910188.57281.188910212.65281.5099
10216.09283.297410226.41294.479210233.29299.108810240.17 302.77110250.96306.0764
#Mann= 3 , 0 , 0
9749.015    0.12       09749.015    0.12       010250.96    0.12       0
#XS Ineff= 2 , 0
       0                               0
Bank Sta=9749.015,10250.96
Exp/Cntr=0.3,0.1

Type RM Length L Ch R = 1 ,10599.82,95.653400,95.653400,95.653400
XS GIS Cut Line= 6
1187988.65817306844382.9351714131187930.58368116844195.558323363
1187916.63018493844143.5758015891187916.14511363844141.635516602
1187897.08994198844072.428686173 1187840.7323977843903.380473446
#Sta/Elev= 30
9749.007296.15039756.768294.4491 9794.55291.3942 9808.29 285.5339832.333272.8661
9870.116269.4815 9880.42265.9376 9887.29261.54079890.725260.64259918.203259.9667
9921.638258.80079931.942252.19059935.377251.40619979.646245.884210000.02241.4722
10020.43243.492210047.66242.348410057.87242.975710071.48247.883810092.21259.3856
10123.33261.690610144.08266.965210168.29 270.75110182.12277.391610220.17280.1969
10223.62283.029610233.26296.429310237.46300.707710244.37304.531610250.98305.6211
#Mann= 3 , 0 , 0
9749.007    0.09       09749.007    0.09       010250.98    0.09       0
#XS Ineff= 2 , 0
       0                               0
Bank Sta=9749.007,10250.98
Exp/Cntr=0.3,0.1

Type RM Length L Ch R = 1 ,10504.17,95.653400,95.653400,95.653400
XS GIS Cut Line= 6
 1188086.9752625844352.6846861631188019.84494411844146.859366236
1188007.73331452844115.6426744041187995.65246981844085.533697269
1187955.72361907843968.7225929131187921.64421663 843878.87197964
#Sta/Elev= 30
 9749.02281.21039766.409279.75059783.664273.30959790.566268.99819800.919260.3023
9804.369258.68319849.231255.82069876.839250.81179900.821250.44469904.446247.7108
9925.152241.0915 9956.21239.74589987.698234.851910001.81234.049710031.44237.2586
 10050.9237.9272 10071.7240.706910078.64242.588510106.37252.914510130.64254.4587
10144.51258.651610154.89260.446710172.46260.671110175.97261.6115   10190269.5575
10207.55269.788110225.09271.312310232.11273.870910246.15288.859310250.99 292.983
#Mann= 3 , 0 , 0
 9749.02    0.12       0 9749.02    0.12       010250.99    0.12       0
#XS Ineff= 2 , 0
       0                               0
Bank Sta=9749.02,10250.99
Exp/Cntr=0.3,0.1

Type RM Length L Ch R = 1 ,10408.51,95.653400,95.653400,95.653400
XS GIS Cut Line= 6
1188182.57323137844332.1958084361188122.26163445844171.797100173
1188089.95015934844055.0789434221188077.96857021 844018.55261612
1188049.83846771843949.1219016241188010.14173978843861.605991828
#Sta/Elev= 30
9749.011280.2915  9769.4275.55699786.994267.17499797.551259.88889804.589257.8261
9822.184256.29419843.297253.20939864.259247.57689882.646247.73319892.329246.9655
9902.011245.30279920.053240.64869950.962237.93329988.397230.855710008.75229.8387
10018.91230.203310077.19236.072610087.74238.889410108.97247.953810123.13251.9408
10147.91253.960210187.42259.976310191.02261.037410198.23265.908710205.43269.5645
10210.69270.281310223.44269.660510245.06271.227410248.66273.064210250.97275.1572
#Mann= 3 , 0 , 0
9749.011  0.1051       09749.011  0.1051       010250.97  0.1051       0
#XS Ineff= 2 , 0
       0                               0
Bank Sta=9749.011,10250.97
Exp/Cntr=0.3,0.1

Type RM Length L Ch R = 1 ,10312.86,95.653400,95.653400,95.653400
XS GIS Cut Line= 6
1188309.81260561844271.0097852411188233.42691384844125.148248728
1188204.24648301844078.6790270541188168.24717071844030.568803489
1188140.20922665 843987.625199591188057.94016339843837.718408247
#Sta/Elev= 30
9749.031270.58749756.904267.03649771.589257.62319778.932254.68949819.315250.7659
9822.987250.15239835.965245.20189845.187 244.2469865.838244.50259882.603237.5578
9886.312236.90419916.367237.03749931.863235.7347 9947.36232.92569970.711 226.947
9999.274226.423410039.87227.989710071.22233.565810090.29241.866110098.02250.5162
 10101.8251.944410124.53254.981210139.67255.594610173.17263.3873 10180.6264.1831
10188.04266.509510202.92275.020110240.51275.220910243.83276.001710250.98 281.951
#Mann= 3 , 0 , 0
9749.031  0.0837       09749.031  0.0837       010250.98  0.0837       0
#XS Ineff= 2 , 0
       0                               0
Bank Sta=9749.031,10250.98
Exp/Cntr=0.3,0.1

Type RM Length L Ch R = 1 ,10217.21,95.653500,95.653500,95.653500
XS GIS Cut Line= 6
1188383.92582598844209.2124119921188335.36354152844123.559818216
1188267.80270653844011.6348055521188257.66523457843991.245967945
1188238.74649001843955.6700118091188127.73446258843777.806429553
#Sta/Elev= 30
9749.025252.18339761.382248.77389791.675246.38029818.076237.80359825.618237.0464
 9848.26237.03779855.924234.81469863.588231.35839909.575229.95379940.233 224.226
9955.768224.2069  9985.9222.61459996.079 219.57510045.27228.041310060.74231.6385
10080.08237.791710107.15251.303310126.49254.318910149.69260.370510165.16266.8922
10176.76270.8418 10184.5275.716110212.36275.533510223.17276.416910227.04278.0818
10230.91281.685610234.78290.768310238.64298.744610242.51303.998410250.96308.5808
#Mann= 3 , 0 , 0
9749.025  0.1037       09749.025  0.1037       010250.96  0.1037       0
#XS Ineff= 2 , 0
       0                               0
Bank Sta=9749.025,10250.96
Exp/Cntr=0.3,0.1

Type RM Length L Ch R = 1 ,10121.55,95.653400,95.653400,95.653400
XS GIS Cut Line= 6
1188475.47889933844163.8260068121188430.55750533844089.629624746
1188352.73607997843968.0489984781188342.38508439 843949.89114674
1188323.45229782843918.3024400421188202.77847667843742.603076141
#Sta/Elev= 30
9749.009250.1092  9758.5245.21019770.006238.21559772.847237.4582 9817.19237.1599
9831.371 235.5969836.176 234.3189842.262231.41779850.779230.37359870.256230.0798
9890.948226.30939928.686225.18159944.268222.85429963.745217.731310005.85215.6699
10009.67215.765110024.97219.225910040.37220.745610084.15230.677810088.13232.0371
10108.03243.758410119.97249.380410127.93 249.95210139.87253.283610151.82254.5049
 10195.6266.335510211.52 274.80410243.36275.339710248.91276.155710250.98277.8398
#Mann= 3 , 0 , 0
9749.009    0.12       09749.009    0.12       010250.98    0.12       0
#XS Ineff= 2 , 0
       0                               0
Bank Sta=9749.009,10250.98
Exp/Cntr=0.3,0.1

Type RM Length L Ch R = 1 , 10025.9,95.653400,95.653400,95.653400
XS GIS Cut Line= 6
1188571.04059818844090.225535758 1188526.9740392844021.854378399
1188478.25911999843956.198420346 1188445.2850322843918.590464721
1188356.47468277843829.7318613671188256.23747326843701.108072961
#Sta/Elev= 30
9749.054236.49319768.732234.98689780.441231.27169790.782 231.4599802.894230.6162
9835.306228.07199867.988224.43959887.982224.26969904.756223.19029926.069220.3473
9955.001217.96319979.769214.20179993.938213.056810008.27213.531310022.62218.2011
10036.97220.148610086.26230.914110090.58232.326110105.97240.085710115.99246.8397
10120.23248.248310132.93248.615810158.34254.036510187.37262.559610201.11264.7711
10212.11265.480810215.98268.502110220.06274.631910228.62275.834210250.97276.1014
#Mann= 3 , 0 , 0
9749.054  0.0756       09749.054  0.0756       010250.97  0.0756       0
#XS Ineff= 2 , 0
       0                               0
Bank Sta=9749.054,10250.97
Exp/Cntr=0.3,0.1

Type RM Length L Ch R = 1 ,9930.246,95.653400,95.653400,95.653400
XS GIS Cut Line= 6
1188631.97248541844032.4124388441188589.45660183843963.382213948
1188553.02345044 843911.014689281188474.89031245843812.170678561
1188389.67186234843712.0605609211188329.91077984843632.383617604
#Sta/Elev= 30
9749.035227.48779754.506226.00289762.212225.43189789.185225.64149812.304224.7438
 9820.01223.62459823.863221.52939827.002220.71169835.621219.47799896.004218.5848
9920.802214.88979943.448215.30769962.717214.73889987.866 211.83410001.58210.9596
10016.96211.8427 10043.1220.260610072.85225.497810093.72231.955110107.32237.8875
10120.25 240.50410128.87241.2436 10146.1240.315210158.66241.857210166.86243.7357
10179.16247.659610209.38261.071610216.07263.331510228.38265.412210250.97264.9345
#Mann= 3 , 0 , 0
9749.035   0.085       09749.035   0.085       010250.97   0.085       0
#XS Ineff= 2 , 0
       0                               0
Bank Sta=9749.035,10250.97
Exp/Cntr=0.3,0.1

Type RM Length L Ch R = 1 ,9834.592,95.653400,95.653400,95.653400
XS GIS Cut Line= 6
1188677.48734083843974.2571681231188613.39997392843853.935070552
1188583.58848297843802.1829244641188550.91331243843756.828307296
1188509.26913412843699.7368846081188412.46856876 843548.80123995
#Sta/Elev= 30
9749.049230.70679773.932225.68169788.801220.8799 9803.67218.87749825.973218.7777
9859.428216.24369863.145216.5645 9877.01216.18729881.731214.88269889.236211.6793
9896.808210.54879923.507209.51689938.457210.33169958.239208.50819993.904206.6028
10023.02207.732710031.14209.165910044.18214.156610059.56215.126210091.23227.4855
10114.62232.362310153.59234.059110169.18236.324810184.77239.421510204.26239.7643
10211.82237.994910219.85237.259410227.65236.909610243.24237.235610250.98236.5837
#Mann= 3 , 0 , 0
9749.049  0.1068       09749.049  0.1068       010250.98  0.1068       0
#XS Ineff= 2 , 0
       0                               0
Bank Sta=9749.049,10250.98
Exp/Cntr=0.3,0.1

Type RM Length L Ch R = 1 ,9738.939,95.653400,95.653400,95.653400
XS GIS Cut Line= 6
1188722.77264824843969.2426025471188661.21148249843827.711110378
1188647.81497511843778.5591997991188624.11133544843638.727709467
1188598.31895813843569.6969721651188562.95055337843497.172717328
#Sta/Elev= 30
9749.096237.0532 9771.44235.92489781.064234.4487 9789.56231.43899804.056 222.926
9811.303221.02629836.548219.60099853.428219.4137 9871.84216.53539893.015 216.326
 9897.94 215.283    9907210.40889937.605209.51399957.912207.65739971.145205.2243
9997.612203.935410024.03204.249210047.34208.048210081.07211.113410115.28 217.294
10132.69225.258310143.29229.052210154.42235.081310160.97237.653210175.27240.6326
10197.18241.385910208.13 242.84410237.33252.369810248.28256.666410250.91258.2774
#Mann= 3 , 0 , 0
9749.096    0.12       09749.096    0.12       010250.91    0.12       0
#XS Ineff= 2 , 0
       0                               0
Bank Sta=9749.096,10250.91
Exp/Cntr=0.3,0.1

Type RM Length L Ch R = 1 ,9643.286,95.653400,95.653400,95.653400
XS GIS Cut Line= 6
1188823.76723013843952.230196917 1188768.1800332843818.402909293
1188724.38691654843677.5367405841188695.27737613843595.918340393
1188672.40041191843541.5107767511188644.22497852843484.300236609
#Sta/Elev= 30
 9749.02247.92549752.532247.53099770.445241.32899797.383238.70589805.551237.2174
9820.601231.5489 9831.33226.30299848.239221.38969873.534219.01179891.119214.9972
9898.088214.17289918.863214.05849925.787211.5746 9929.25208.53829932.712206.6733
9936.175206.06439977.446204.15549997.921201.242210049.37203.041710108.58210.2128
   10126214.630110143.75222.9395 10165.1 227.639 10182.9233.466410201.07236.8941
10212.04241.306910233.98241.142810237.64242.362610244.95247.207910250.97250.0396
#Mann= 3 , 0 , 0
 9749.02  0.0999       0 9749.02  0.0999       010250.97  0.0999       0
#XS Ineff= 2 , 0
       0                               0
Bank Sta=9749.02,10250.97
Exp/Cntr=0.3,0.1

Type RM Length L Ch R = 1 ,9547.632,93.262100,93.262100,93.262100
XS GIS Cut Line= 6
1189034.99547174 844128.314412531188905.56763974843880.455287453
1188800.70411864 843619.282846061188753.88209915843519.834120588
1188670.74645149843382.5148052341188570.27074045843245.291701157
#Sta/Elev= 30
9499.028252.03179512.659252.64779531.327261.52489562.975267.2986 9617.96266.2607
9647.071256.46119676.591253.81349688.801248.26799731.492247.21769757.112 237.738
9793.606236.25579807.814231.42629832.969216.10779879.407213.67539922.013208.4799
9932.664204.35379995.761198.621110090.84203.538910152.77 214.65910201.14229.9393
10216.22231.447710235.08243.716910258.01252.980610278.01 253.33310320.44262.9097
10355.28276.5342 10416.8278.054210449.65293.522310477.25295.672810500.96309.9556
#Mann= 3 , 0 , 0
9499.028  0.0796       09499.028  0.0796       010500.96  0.0796       0
#XS Ineff= 2 , 0
       0                               0
Bank Sta=9499.028,10500.96
Exp/Cntr=0.3,0.1

Type RM Length L Ch R = 1 , 9454.37,93.262000,93.262000,93.262000
XS GIS Cut Line= 6
1189087.91033683 844004.366437311188963.21933482843776.289253505
1188895.42316497843607.0324794851188870.74877011 843557.89148823
1188800.57463736843448.832457612 1188695.3621449843309.356716529
#Sta/Elev= 30
9599.047236.19699662.719238.69679689.137235.95429738.199235.60349764.116231.6755
 9786.32226.03639823.326 213.6149838.129211.71229874.704209.74449885.508204.7604
9892.711203.52019917.921 203.8349932.327200.92929974.417198.96529998.789196.2248
10040.68195.775910088.36197.695410126.39202.521610166.59203.618910172.99205.5319
10195.97218.1316 10216.5225.781610240.59227.816410260.87241.022410275.58246.7555
10305.61249.924810322.21250.259710347.12253.855410356.93253.648410400.94263.0551
#Mann= 3 , 0 , 0
9599.047  0.1007       09599.047  0.1007       010400.94  0.1007       0
#XS Ineff= 2 , 0
       0                               0
Bank Sta=9599.047,10400.94
Exp/Cntr=0.3,0.1

Type RM Length L Ch R = 1 ,9361.108,93.262100,93.262100,93.262100
XS GIS Cut Line= 6
1189227.55375521843919.557071535 1189042.5252945843653.826158709
1189013.85351475843622.0812929491188961.90492137843581.798792938
1188932.94394385843552.3316908561188726.24789929843297.435551419
#Sta/Elev= 30
9599.081215.27469623.052214.36519634.995211.99479656.983210.62459691.738210.3749
9709.115206.42579755.455206.11729772.833204.7218 9786.27201.95899830.061200.6197
9859.641197.56359882.337198.29969894.541197.30599940.709197.13759998.652193.9663
10089.89193.875410115.96197.4015   10136202.312310179.21203.683210182.11204.3633
 10190.5212.182310194.69214.230310242.47 223.53710273.46233.7051 10304.3238.9097
10319.72245.733310342.96249.303710372.79251.422710386.53256.704810400.93258.1031
#Mann= 3 , 0 , 0
9599.081  0.1157       09599.081  0.1157       010400.93  0.1157       0
#XS Ineff= 2 , 0
       0                               0
Bank Sta=9599.081,10400.93
Exp/Cntr=0.3,0.1

Type RM Length L Ch R = 1 ,9267.846,109.942200,109.942200,109.942200
XS GIS Cut Line= 6
1189277.44890716843865.9201295781189079.61893613843600.204491038
1189056.94317676843560.4535055011189037.11399909843502.126738891
1189014.01032336843467.0023995861188781.66649794843245.717351459
#Sta/Elev= 30
 9599.05214.36869638.336211.48929659.316207.11319720.926203.68739737.355199.8049
9766.106199.09969778.428197.86889786.643198.53199807.388198.09029831.823195.7523
9856.465196.18759868.564195.14439908.895194.42699935.933191.48649967.189 192.957
10012.45190.882910040.82191.948610084.84195.486510125.67196.911810197.76204.1764
10238.15213.901510250.78  215.0210264.03214.658610282.02 218.30510309.55225.5088
10318.73227.1282 10332.5232.378310342.88  235.3210380.42242.477610400.91249.1107
#Mann= 3 , 0 , 0
 9599.05  0.1057       0 9599.05  0.1057       010400.91  0.1057       0
#XS Ineff= 2 , 0
       0                               0
Bank Sta=9599.05,10400.91
Exp/Cntr=0.3,0.1

Type RM Length L Ch R = 1 ,9157.904,150.926800,150.926800,150.926800
XS GIS Cut Line= 6
1189416.29544716843777.2131229321189305.88403912843654.769824947
1189169.85264728843517.5722260511189122.90878359843460.086052779
1188962.40244636843346.9596271471188831.50863504843233.891509337
#Sta/Elev= 30
9603.395208.89069623.643199.65749641.117197.19329848.277194.02249879.516195.5778
9945.299192.43159997.645188.753210017.92191.451210026.72191.568410040.42 189.089
10046.16189.367810085.29194.676810108.94192.413610116.83194.586810128.65194.2247
10156.24197.346910176.19200.238810190.38204.052910224.87205.255810245.18209.5991
10276.26212.196510286.63216.191410302.17218.497910313.56221.797810322.06222.9539
10342.25229.115210356.83230.346610376.28235.345210388.76236.374910405.29239.3382
#Mann= 3 , 0 , 0
9603.395  0.1129       09603.395  0.1129       010405.29  0.1129       0
#XS Ineff= 2 , 0
       0                               0
Bank Sta=9603.395,10405.29
Exp/Cntr=0.3,0.1

Type RM Length L Ch R = 1 ,9006.977,112.179300,112.179300,112.179300
XS GIS Cut Line= 6
1189595.33218998843709.0415901691189374.00451317843465.022250965
 1189292.4231765843409.7077147221189172.87541175843359.058166668
1189019.80501679843272.5986851011188826.40619382843120.306479827
#Sta/Elev= 30
9417.802208.41399447.593206.65319473.321197.79929483.329195.8851  9573.6193.3806
9663.473193.17959673.537191.78279719.282191.48589747.761193.13849762.533191.5644
9810.834191.2549  9850.9184.86279882.037186.08129938.729184.49759966.937186.0884
9997.607183.648810028.82185.798210083.85196.622910098.53200.9703 10131.5203.8964
10151.25213.040310190.49221.404110215.91  224.2310232.29230.432910270.51239.4629
10285.93245.2941 10296.2251.331510340.66252.165810356.63265.7673   10399 285.533
#Mann= 3 , 0 , 0
9417.802    0.12       09417.802    0.12       0   10399    0.12       0
#XS Ineff= 2 , 0
       09869.987                       0
Bank Sta=9417.802,10399
Exp/Cntr=0.3,0.1

Type RM Length L Ch R = 1 ,8894.798,93.262100,93.262100,93.262100
XS GIS Cut Line= 6
 1189633.5266344843679.5277012881189447.86797145843447.906370729
1189385.08420321  843391.44721591189257.43737236843286.482218131
1189103.90010393843168.6210841241188899.87755314   842986.309974
#Sta/Elev= 30
9387.198209.32159416.044207.11899438.274195.66149445.477193.23079529.572192.2592
 9634.69193.0726 9714.77188.91389758.929188.97669799.748185.24389835.907184.8783
9857.728187.3662 9925.69181.643910003.73181.387210028.19182.772510049.69187.3017
10070.59193.4841 10090.7201.363910146.05226.759110168.09233.638710198.13 248.135
 10211.2251.543310218.16255.013510268.14255.944910281.48257.512110296.79270.0073
10325.94288.931210339.28291.901410359.99294.0423 10384.3305.987810400.98316.3632
#Mann= 3 , 0 , 0
9387.198  0.0942       09387.198  0.0942       010400.98  0.0942       0
#XS Ineff= 2 , 0
       09852.891                       0
Bank Sta=9387.198,10400.98
Exp/Cntr=0.3,0.1

Type RM Length L Ch R = 1 ,8801.536,193.432500,193.432500,193.432500
XS GIS Cut Line= 6
1189682.13774553843650.0138124081189347.66506711843300.398647547
1189310.08237341843251.2727877351189187.36353409843053.519715071
1189082.82516909842935.8525504321188956.13359964842812.877069101
#Sta/Elev= 30
9387.979 210.8779409.792206.44379427.729198.86049445.666193.65429694.692 190.995
9709.922188.62669747.188186.56719819.359187.00889831.533188.24819875.006187.4843
9910.977182.64219995.248177.821310008.14178.747710036.62184.023310071.95194.0942
10127.54214.931910158.89229.047910180.04234.014410201.54243.843310216.36247.4256
10266.97264.032410294.86277.523110339.08292.731910365.73305.321410398.16313.3264
10418.45316.052910447.88 327.89310475.01328.675810493.09332.342510500.93332.5068
#Mann= 3 , 0 , 0
9387.979    0.12       09387.979    0.12       010500.93    0.12       0
#XS Ineff= 2 , 0
       09859.869                       0
Bank Sta=9387.979,10500.93
Exp/Cntr=0.3,0.1

Type RM Length L Ch R = 1 ,8608.103,193.432400,193.432400,193.432400
XS GIS Cut Line= 6
1189733.08251444843493.0059760921189560.50077152843283.844777371
1189387.04312316843009.1520814551189312.99829028842904.768831255
1189222.84915172842803.4138267781189118.42691482842707.270631622
#Sta/Elev= 30
9499.059203.10539520.795196.63669542.494193.55259620.611189.79169655.194184.3505
9746.102182.21779763.091 184.1169814.795 180.9289838.499184.53669908.624178.7819
9966.199177.92949981.552178.673310000.79174.970810008.52176.0302 10020.1181.5445
10050.98183.244610074.15186.120910176.98 206.17310196.17209.220910239.22213.3761
10260.68217.988110273.55221.309210290.72227.609710312.99233.094410323.48237.8851
10333.03239.209710353.65245.798710438.98275.272810473.56285.595310500.95291.8901
#Mann= 3 , 0 , 0
9499.059  0.1102       09499.059  0.1102       010500.95  0.1102       0
#XS Ineff= 2 , 0
       0                               0
Bank Sta=9499.059,10500.95
Exp/Cntr=0.3,0.1

Type RM Length L Ch R = 1 ,8414.671,193.432500,193.432500,193.432500
XS GIS Cut Line= 6
1189919.49708163843411.7794586191189716.28005229843181.294835124
1189560.92363554842936.5390147921189506.82071528 842863.85783967
 1189405.1636617842762.5289273191189271.47926172842657.418747692
#Sta/Elev= 30
9499.049208.05459527.504205.23329536.609202.24749581.953193.10779618.057192.2892
9647.233188.51999670.852187.64879692.399185.63619760.761183.16719785.726184.1168
 9838.42178.60569866.323179.55229917.562175.36139959.604174.1684  9987.7171.7429
10017.12172.619710051.82177.421710075.35177.745110090.37179.599210106.14179.8679
10126.15 181.85610167.31187.855810228.31198.502310279.59 210.015 10361.2231.4056
10382.49238.643810437.59253.962710448.43258.083310480.98267.941810500.93271.6344
#Mann= 3 , 0 , 0
9499.049  0.1144       09499.049  0.1144       010500.93  0.1144       0
#XS Ineff= 2 , 0
       0                               0
Bank Sta=9499.049,10500.93
Exp/Cntr=0.3,0.1

Type RM Length L Ch R = 1 ,8221.238,193.432400,193.432400,193.432400
XS GIS Cut Line= 6
1190129.65682412843243.5821871161189824.04701121842994.498138309
1189776.72187506842942.767636171  1189735.459043842872.075254538
1189699.23859381842836.3823225891189351.09409894842630.912204431
#Sta/Elev= 30
9499.048194.04969541.158192.84579583.353189.50299599.176187.32629612.003186.8422
9637.144188.46769657.195187.59079674.855185.68629699.996185.04489729.327181.6146
9805.506176.41039831.099176.75439857.384 174.8739902.946174.31279976.373171.8336
10013.73172.664910032.61173.881510064.17173.052710082.49174.626110135.13176.4788
10180.49183.577410225.56192.045310278.14 203.91510308.19210.961210342.42 220.026
10350.14221.214110442.07  244.69 10480.4253.3854 10491.9257.2515 10500.9257.9301
#Mann= 3 , 0 , 0
9499.048    0.12       09499.048    0.12       0 10500.9    0.12       0
#XS Ineff= 2 , 0
       0                               0
Bank Sta=9499.048,10500.9
Exp/Cntr=0.3,0.1

Type RM Length L Ch R = 1 ,8027.806,193.432500,193.432500,193.432500
XS GIS Cut Line= 6
1190278.39452115842819.4540110371190105.41457608842754.833743284
1189950.69919299842722.0780676631189656.71764461842745.447670285
1189532.01222366842700.7004353061189331.89214681842592.969184127
#Sta/Elev= 30
9499.151 189.5689609.655190.4562 9678.94192.79269723.253 192.7069770.461189.3272
9783.822185.44139813.708179.90149830.311179.71929883.009172.18069902.726170.8964
9925.738170.77549965.632173.07739992.955172.0654 10020.6 173.32910044.26172.0669
10054.23 173.28510074.07172.225810083.91173.798310110.22180.320410153.68184.4102
10212.32197.440110254.98209.030310324.11224.1782 10360.8234.250310383.34238.5889
10436.06251.740910462.41253.536910473.71257.651410488.77259.010510500.83261.3739
#Mann= 3 , 0 , 0
9499.151    0.12       09499.151    0.12       010500.83    0.12       0
#XS Ineff= 2 , 0
       0                               0
Bank Sta=9499.151,10500.83
Exp/Cntr=0.3,0.1

Type RM Length L Ch R = 1 ,7834.373,193.432400,193.432400,193.432400
XS GIS Cut Line= 6
1190286.95396796842664.2215112061190061.40101106842595.168398619
1189735.66438756842535.6004698551189579.66080046842499.963197692
1189448.65512665842458.1340755361189321.69729393842406.416598327
#Sta/Elev= 30
9499.036 203.8369575.294205.8775 9609.79207.77479654.145207.52829681.301206.1293
9725.429201.18579773.392191.53059789.193 187.524 9802.59186.07589812.638183.3272
9862.681182.03169875.996 177.3539895.968171.86679899.297 171.8379912.612 174.142
9925.927172.78279952.557172.18889992.502172.015410029.16172.930210052.49171.2329
10055.82171.602510065.83175.045210082.59176.854410109.42184.211210264.59220.9898
10292.44225.917610337.44 225.81310351.33226.7599 10393.4225.838310500.97217.8565
#Mann= 3 , 0 , 0
9499.036   0.049       09499.036   0.049       010500.97   0.049       0
#XS Ineff= 2 , 0
       0                               0
Bank Sta=9499.036,10500.97
Exp/Cntr=0.3,0.1

Type RM Length L Ch R = 1 ,7640.941,193.432500,193.432500,193.432500
XS GIS Cut Line= 6
1190325.61076832842503.5003108541190261.01575861842479.470641469
1190162.18303839842447.1814847941189556.13261048842278.911628347
1189461.32798174 842249.491222821189366.23680576842215.996903662
#Sta/Elev= 30
9499.027224.06159588.641229.8642 9633.51229.56519647.316223.18299671.477218.9113
9681.697215.97749705.531205.29779760.761190.43689770.222186.82089790.651183.4921
9800.865180.05659841.723177.23899865.557171.11269906.414171.72049913.224175.2703
9920.033177.15889943.867178.88319971.106173.015610076.67 171.463 10097.1175.5982
10117.53182.281110141.36187.5444 10168.6192.114610209.46195.161410274.16193.6139
10356.37185.210810394.15183.6612 10421.9179.718410479.01186.026410500.98190.1336
#Mann= 3 , 0 , 0
9499.027  0.0467       09499.027  0.0467       010500.98  0.0467       0
#XS Ineff= 2 , 0
       0                10205.73       0
Bank Sta=9499.027,10500.98
Exp/Cntr=0.3,0.1

Type RM Length L Ch R = 1 ,7447.508,168.433800,168.433800,168.433800
XS GIS Cut Line= 6
1190373.32845148842312.4844695931190246.36956003842260.759861767
1190096.03423211842212.1570326831189822.17702186842162.401239872
1189630.07047024 842120.446970851189140.47107887841962.513812393
#Sta/Elev= 30
9499.029213.57439549.811218.36159567.556 215.3479609.829217.76559683.093199.4723
9707.383189.47849745.283181.43329776.073182.99799806.718171.62799823.628173.7729
10076.93173.389410100.36171.563610143.89178.2256 10214.3181.328710258.25179.5305
10322.92170.930510398.31172.195410412.07170.448610437.19173.381810456.95172.2505
10470.78174.678910488.08173.528610560.71178.079810633.35184.663910643.73183.6004
10661.03 187.592 10688.7   186.610740.58193.021410754.42191.182410783.98193.9459
#Mann= 3 , 0 , 0
9499.029  0.0508       09499.029  0.0508       010783.98  0.0508       0
#XS Ineff= 2 , 0
       09798.035        10174.02       0
Bank Sta=9499.029,10783.98
Exp/Cntr=0.3,0.1

Type RM Length L Ch R = 1 ,7279.075,144.871700,144.871700,144.871700
XS GIS Cut Line= 6
1190376.26791288842181.0123518181190221.67958697842106.930021512
1190059.57008907842042.0555680711189969.06563254842014.777751778
1189749.67170846841969.8519955191189432.42818344841856.366876215
#Sta/Elev= 30
9503.133205.6474 9543.82 200.6969563.354197.01689580.394195.90959605.995189.4311
 9616.85187.77429631.507182.15799685.289180.28419706.682177.1758 9724.51 171.382
9728.075171.04699749.468172.31459830.252 172.787 9882.34172.15489980.561173.5905
10117.44171.814810171.91172.554310185.66171.805610195.97173.049110223.46172.5203
10244.09174.597710268.37172.103210275.31 172.34710285.71174.527310299.59172.6191
10313.46176.964410344.89 180.614 10376.4185.721610428.93195.800110505.06 207.072
#Mann= 3 , 0 , 0
9503.133  0.0414       09503.133  0.0414       010505.06  0.0414       0
#XS Ineff= 2 , 0
       09806.928        10142.29       0
Bank Sta=9503.133,10505.06
Exp/Cntr=0.3,0.1

Type RM Length L Ch R = 1 ,7134.203,73.559400,73.559400,73.559400
XS GIS Cut Line= 3
1190341.85996777 842096.194367961190263.73496777842031.958256871
1189650.88774553841707.305479065
#Sta/Elev= 30
9558.267189.50579585.436185.13249606.099181.16769628.932179.28799637.427175.3775
9657.757171.66439662.471171.30499673.609172.2649 9688.46172.70759703.311174.3148
9721.875173.10019736.726172.63649832.382172.88019874.098172.16759900.087172.8224
 9944.64171.67439978.055172.530810011.47172.7876 10137.7171.118510171.12171.6793
10197.11174.771310231.87181.022610267.65189.006210280.93191.159410293.64193.9746
10301.96195.282210322.98200.172110330.77201.4099 10341.9204.501910352.94206.4215
#Mann= 3 , 0 , 0
9558.267  0.0527       09558.267  0.0527       010352.94  0.0527       0
#XS Ineff= 2 , 0
       09840.203        10114.71       0
Bank Sta=9558.267,10352.94
Exp/Cntr=0.3,0.1

Type RM Length L Ch R = 1 ,7060.644,67.402200,67.402200,67.402200
XS GIS Cut Line= 6
1190454.10281581842127.0332522551190349.57099531842044.742244602
1190306.20141018 841961.339196311190069.33675305  841841.2388068
1189952.57248542841788.972896517  1189682.346609841657.752100543
#Sta/Elev= 30
9437.192225.33689449.087226.37039457.438225.11799469.964218.72969495.017203.8935
9504.336199.94359514.944194.07299528.421191.07969540.948184.54089583.455182.1948
9594.549175.92059605.642173.39549619.919175.62389685.453174.8729  9723.4178.1166
9736.951177.67919747.987178.29089832.221176.05789873.055172.85349898.804171.8493
9912.024169.76399931.862169.038410065.02170.215710171.55174.048810233.29 181.573
10271.11189.8651 10291.4196.017910327.71197.728210338.61198.962210358.16202.9814
#Mann= 3 , 0 , 0
9437.192    0.12       09437.192    0.12       010358.16    0.12       0
#XS Ineff= 2 , 0
       09886.673        10121.86       0
Bank Sta=9437.192,10358.16
Exp/Cntr=0.3,0.1

Type RM Length L Ch R = 1 ,6993.241,195.360600,195.360600,195.360600
XS GIS Cut Line= 2
1190179.21709985841835.680130631 1189827.8184984841632.866740301
#Sta/Elev= 30
9845.759167.65359857.931168.28929868.728167.89559876.304166.9137 9897.31166.5648
9899.032166.29759921.761158.25399936.913154.28399959.641151.88829974.794151.9975
 9995.76154.886610001.31155.251110008.89 155.07710020.25153.735910031.61154.3089
10042.98 152.71710092.22155.938510100.77157.678910111.16160.899310120.46165.8183
10127.03167.994810137.68173.148910146.72176.329410156.62178.534510190.71180.6451
10199.22180.062210209.65178.204910217.23177.558910239.96177.756910251.49179.4534
#Mann= 3 , 0 , 0
9845.759    0.12       09845.759    0.12       010251.49    0.12       0
#XS Ineff= 2 , 0
       0                               0
Bank Sta=9845.759,10251.49
Exp/Cntr=0.3,0.1

Type RM Length L Ch R = 1 ,6797.881,195.360700,195.360700,195.360700
XS GIS Cut Line= 6
1190538.17743111841892.3481738911190284.19800695841680.572960962
1190225.34270878841636.2013183571190178.15795773841607.938398699
1190047.18191404841542.6734497011189711.41353227 841332.68572718
#Sta/Elev= 30
9499.075183.45429567.478  186.489589.761181.07239614.284172.07539619.473171.1249
9696.826171.62299765.583170.88299778.476164.17469781.916163.49469827.634162.4263
9854.727151.78069865.627149.31099892.876148.45859903.486148.98829938.374145.2983
9979.267 142.58910008.16143.830710033.41143.687710085.52148.410610104.24152.5306
 10143.1155.211710170.32158.2589 10236.6160.280710271.42163.046310318.09168.7545
10341.42169.227310391.47172.850910422.18177.2219 10479.1179.340810500.96182.7191
#Mann= 3 , 0 , 0
9499.075    0.12       09499.075    0.12       010500.96    0.12       0
#XS Ineff= 2 , 0
       0                               0
Bank Sta=9499.075,10500.96
Exp/Cntr=0.3,0.1

Type RM Length L Ch R = 1 , 6602.52,195.360600,195.360600,195.360600
XS GIS Cut Line= 6
1190613.55377805841830.2839598781190505.04723118841733.068171041
1190414.12190914 841640.151591921190215.31620054841377.202158318
1190163.01963731841317.9700855961190016.00244631841196.397978604
#Sta/Elev= 30
9499.082180.80839564.029178.79499597.973 164.1569618.112159.69349628.808159.0782
9646.497155.96419692.386158.66699734.943167.67759748.892  168.479771.447166.2398
9780.145163.07989831.182  161.339866.682151.17629892.707147.20299912.955146.4809
9940.512143.37799956.446139.287210010.68138.758810027.77140.883310038.81143.6847
 10056.2152.547510105.04169.727410135.95 183.45610170.57186.671510197.82192.7983
10217.54194.507610231.91198.733210282.75208.7175 10306.5211.379510374.75222.8835
#Mann= 3 , 0 , 0
9499.082    0.12       09499.082    0.12       010374.75    0.12       0
#XS Ineff= 2 , 0
       0                               0
Bank Sta=9499.082,10374.75
Exp/Cntr=0.3,0.1

Type RM Length L Ch R = 1 ,6407.159,195.360700,195.360700,195.360700
XS GIS Cut Line= 6
1190817.17253196  841706.83916311190637.74324347841546.249958598
1190460.44095451841379.2549969391190352.98295954841282.224134885
1190281.78011631841225.5126781821190147.76472084 841129.75078161
#Sta/Elev= 30
9499.014181.4016 9677.39180.38559698.666178.50079728.183173.34959770.561167.7194
9795.492174.06599806.617172.52839815.631174.39849833.773173.84549862.484170.5359
9901.263  141.77 9905.77140.97799928.304141.72089955.346138.17839991.209 135.568
10048.64138.925110057.49139.884710070.27143.303110094.72143.628410106.16 145.658
10119.43146.135910136.66150.944410149.25156.074610170.22156.057110203.77164.3716
10268.42182.227710290.61189.558410325.91198.590710369.84  207.7310383.92209.2199
#Mann= 3 , 0 , 0
9499.014    0.12       09499.014    0.12       010383.92    0.12       0
#XS Ineff= 2 , 0
       0                               0
Bank Sta=9499.014,10383.92
Exp/Cntr=0.3,0.1

Type RM Length L Ch R = 1 ,6211.799,195.360600,195.360600,195.360600
XS GIS Cut Line= 6
1190942.55038443841452.984635061 1190786.3084363841322.197680536
1190668.16058606841243.1333957041190586.93139146841207.976745889
1190400.59104807841158.0232344191190243.98480826841081.081318785
#Sta/Elev= 30
9499.085181.91329580.131181.62789597.441180.3456 9642.06 179.864 9686.43176.2677
9711.411176.40969715.929 175.7219731.707 168.2469739.825162.89079743.786 161.916
 9776.24159.58389796.451160.39829827.847159.64359833.958158.54429849.125151.2763
9852.767150.38129869.648150.10559878.266 147.3029889.194146.56319896.381143.8129
 9945.12142.41699995.918132.590410042.99137.358510087.22140.573710104.49145.6859
10128.72151.070710207.54177.582410225.86182.565910255.68 189.50110301.52197.5035
#Mann= 3 , 0 , 0
9499.085  0.0836       09499.085  0.0836       010301.52  0.0836       0
#XS Ineff= 2 , 0
       0                               0
Bank Sta=9499.085,10301.52
Exp/Cntr=0.3,0.1

Type RM Length L Ch R = 1 ,6016.438,195.360600,195.360600,195.360600
XS GIS Cut Line= 6
1190951.20352865841335.7115780561190616.40698368841027.152126887
1190595.99278608841015.003577399 1190551.6471988840997.181505218
1190514.02141787840976.872868627 1190364.3603438 840881.76870677
#Sta/Elev= 30
9499.081 178.1629602.659174.1443 9633.69174.43819637.944173.41899642.556169.9621
9647.701163.5141 9652.58 160.0479695.751158.44679735.516158.47249740.081155.8016
9753.541145.04579758.086143.52359783.247142.61089858.081143.26599878.058142.4683
9882.798141.77059921.618131.55479947.274129.28159985.637131.577710024.53132.1036
10050.54134.450310092.53140.0505 10131.4146.404710150.84150.402210166.38152.2985
10174.16154.222510197.48157.465910216.92 162.19510234.48163.905910246.09166.5509
#Mann= 3 , 0 , 0
9499.081  0.1026       09499.081  0.1026       010246.09  0.1026       0
#XS Ineff= 2 , 0
       0                               0
Bank Sta=9499.081,10246.09
Exp/Cntr=0.3,0.1

Type RM Length L Ch R = 1 ,5821.078,195.360700,195.360700,195.360700
XS GIS Cut Line= 6
1191061.48942811841311.4622316461190930.31306833841184.346282108
1190841.40874589841084.8843792011190643.27340298840781.310376943
1190575.02409162840708.6264470421190532.66888826840673.184297737
#Sta/Elev= 30
9499.045 173.606 9562.18173.87499641.304171.86179649.374170.29169659.945165.9496
9696.666165.79269700.926 162.959 9705.73 157.427 9741.58155.99239794.308157.4906
9798.045155.29139809.571144.42079815.214  142.859946.192142.15549950.066140.6882
9953.941136.5463 9955.23136.12639997.168127.1888 10008.8126.664810059.27129.9203
10074.49  133.6110090.74140.918710103.68144.241410143.44149.460910164.02149.7352
10201.44165.594210242.21179.223910284.52187.048910315.03190.722210332.97191.0797
#Mann= 3 , 0 , 0
9499.045    0.12       09499.045    0.12       010332.97    0.12       0
#XS Ineff= 2 , 0
       0                10315.61       0
Bank Sta=9499.045,10332.97
Exp/Cntr=0.3,0.1

Type RM Length L Ch R = 1 ,5625.717,195.360600,195.360600,195.360600
XS GIS Cut Line= 6
1191256.18493059841145.0440581491191150.24874988841049.266587776
1190946.01518055840855.3790459581190819.64448638840776.303422883
1190685.26858084840662.8828356291190617.54740316840613.957124403
#Sta/Elev= 30
9499.079149.88539575.701 150.3059583.947148.70149593.731143.94569603.515142.5581
9613.299142.32979623.083143.15199660.339142.08439699.151142.25989708.572139.8103
9717.993138.73869812.206138.31989929.577 140.0629934.742138.78169964.717 127.087
9977.805128.68839983.846127.9057    9999123.909210028.46125.238310054.05130.5311
10073.89131.442910082.25134.709310099.01 144.61610107.37147.383510163.55149.6238
10180.01151.088410211.08164.647710224.05167.5674 10289.8168.8886 10332.2 168.394
#Mann= 3 , 0 , 0
9499.079    0.12       09499.079    0.12       0 10332.2    0.12       0
#XS Ineff= 2 , 0
       0                10304.29       0
Bank Sta=9499.079,10332.2
Exp/Cntr=0.3,0.1

Type RM Length L Ch R = 1 ,5430.356,320.896500,320.896500,320.896500
XS GIS Cut Line= 6
1191296.72107884 841096.194367961191085.55025047840777.521440908
1190981.50718832840634.5823862111190939.96989214840596.855635703
1190906.84622383 840577.738590361190847.06830108840557.999923512
#Sta/Elev= 30
9501.033141.90429538.261141.01479550.068140.18639573.683137.55759613.041136.8726
9624.848136.13219644.527 133.7669695.693133.62559703.564131.6513  9707.5 131.195
9790.152 129.5979829.509127.51719837.675126.38749935.762 125.2819971.925126.3247
9979.749125.5092   10001124.720310041.77125.467710055.23126.434910077.45128.8641
10107.97133.004210135.29135.143310154.82136.112610159.35136.828610164.65139.2651
 10168.1 137.34510171.56140.216910181.92146.071110192.29146.958910217.77 147.149
#Mann= 3 , 0 , 0
9501.033  0.0839       09501.033  0.0839       010217.77  0.0839       0
#XS Ineff= 2 , 0
       0 9875.94                       0
Bank Sta=9501.033,10217.77
Exp/Cntr=0.3,0.1

Type RM Length L Ch R = 1 , 5109.46,360.203000,360.203000,360.203000
XS GIS Cut Line= 6
1191716.87130699840240.0362592791191357.87419158840326.394177392
1191269.90757143840346.5031032561191203.11782545840358.139293298
1191135.79183602840387.5071855931190883.37319774840543.204663406
#Sta/Elev= 30
9298.207160.98459334.453156.56129347.286154.07369368.198151.99659401.942146.2886
 9439.06143.36559476.179138.58659536.919135.63929553.791134.39959570.663134.0304
9590.909134.3941 9614.53132.59269641.526128.09459665.147122.51079836.748122.3937
9876.121120.8679 9909.06120.49329955.317120.736310001.57121.819710009.28121.3454
10016.99121.6007 10024.7124.354510032.41125.888610051.69127.737410063.25128.3044
10078.67130.729410132.64134.699110159.62135.4758 10186.6144.9056 10195.5146.7453
#Mann= 3 , 0 , 0
9298.207   0.085       09298.207   0.085       0 10195.5   0.085       0
#XS Ineff= 2 , 0
       0                               0
Bank Sta=9298.207,10195.5
Exp/Cntr=0.3,0.1

Type RM Length L Ch R = 1 ,4749.257,219.047100,219.047100,219.047100
XS GIS Cut Line= 6
1191571.97832714840082.8554786211191243.22711112840120.559755406
1190960.12477686840107.0028018721190889.29791568840108.649536363
1190674.85826175840142.1696281351190205.36853297 840198.90513008
#Sta/Elev= 30
9492.046173.74379527.046178.26759576.679176.71019596.532180.03519613.076180.7615
9679.286175.7052 9712.34169.41189728.836168.48069797.949154.15819814.404148.9475
 9929.29120.14289945.723119.14819952.296117.08659975.302 115.6139998.313112.5493
10011.47113.954410044.37120.366610070.68120.800210126.56115.714110142.97117.5047
10169.22115.483710261.69117.539710274.97116.709610338.28123.163510411.57122.7615
10467.75128.300510494.19 129.72810613.16133.770810659.43133.797210867.51143.9532
#Mann= 3 , 0 , 0
9492.046    0.07       09492.046    0.07       010867.51    0.07       0
#XS Ineff= 2 , 0
       0                               0
Bank Sta=9492.046,10867.51
Exp/Cntr=0.3,0.1

Type RM Length L Ch R = 1 , 4530.21,156.088400,156.088400,156.088400
XS GIS Cut Line= 6
 1191442.1022358 839788.95869829 1191305.3840102839792.361545987
1191193.43457878839818.2859106251191093.00611648839857.657266442
1190834.38460602839990.4403864711190494.20132686840074.814536473
#Sta/Elev= 30
9499.061193.15539591.043184.85619643.926178.73759684.024176.09769714.387 170.842
9758.841166.1593 9814.67162.0466 9836.15158.90979864.952151.71159901.778139.7199
9931.729126.16579958.168119.03049984.608109.13649995.939107.695110044.82112.4297
10063.47 109.41910074.36114.003610092.52118.731210117.56116.990610142.27110.5769
10156.26109.053810180.41117.873610201.12120.477810221.66126.833810228.46127.8714
10252.23124.9312   10276125.479410289.59128.957710327.57133.204610500.95138.8822
#Mann= 3 , 0 , 0
9499.061  0.0881       09499.061  0.0881       010500.95  0.0881       0
#XS Ineff= 2 , 0
       0                               0
Bank Sta=9499.061,10500.95
Exp/Cntr=0.3,0.1

Type RM Length L Ch R = 1 ,4374.121,0.000000,0.000000,0.000000
XS GIS Cut Line= 6
1191401.26312525 839746.756235941191301.95381457 839730.12493153
1191232.71630949839728.8342226881191175.65660984839733.413804733
1190620.39410776839837.1733710461190413.14326308839868.065393221
#Sta/Elev= 30
9508.911 180.8919567.662173.03519607.307165.78319666.386157.24989692.679154.8649
 9719.01151.22689791.906145.24189818.587141.98789848.712136.92959878.838133.8822
9898.922128.9512 9932.04114.26849959.174112.1913 9975.87108.1748 9995.75104.5215
10025.58107.291910035.53110.246310045.48115.420310052.12117.473610209.33122.0785
10242.78125.970710272.89127.525110292.96132.281610329.59133.652310359.51136.8983
10379.46140.272810415.99143.787110429.23143.729610488.81146.793610510.77148.9993
#Mann= 3 , 0 , 0
9508.911  0.0821       09508.911  0.0821       010510.77  0.0821       0
#XS Ineff= 2 , 0
       0                               0
Bank Sta=9508.911,10510.77
Exp/Cntr=0.3,0.1
